HEC-RAS study BIGSPRFK.prj: BIGSPRFK

--- BIGSPRFK.g01 (geometry) --- (continued)

Type RM Length L Ch R = 1 ,23531   ,239.5,242.2,244.4
BEGIN DESCRIPTION:
xs 1
END DESCRIPTION:
XS GIS Cut Line= 3
2238072.77284131 517181.794986542237944.10991265517290.895130733
2237668.72610041  517630.9866147
#Sta/Elev= 30
       0 2900.01    54.7 2896.68   144.7 2894.04   158.1 2894.58   181.9  2893.6
     194 2894.21   274.6 2890.07   336.3 2889.15   366.5 2887.37   377.5 2885.52
   403.8 2884.09   414.9  2884.4   420.5 2885.54   429.1 2886.96   439.3 2894.28
   446.1 2896.75   454.6  2897.1   483.1 2895.36     486 2895.82   490.7 2900.12
   497.3  2907.6   506.2 2924.23   511.8 2932.96   514.4 2935.63   554.2 2962.29
   557.6 2966.02   567.9 2982.66     577 2990.46   583.4 2994.78606.2974 3003.34
#Mann= 5 ,-1,0
       0     .05       0  358.69     .06       0   377.5    .045       0
   420.5     .06       0  488.69      .1       0
Bank Sta=377.5,420.5
XS Rating Curve= 0 ,0
Exp/Cntr(USF)=0,0
Exp/Cntr=0.3,0.1

Type RM Length L Ch R = 1 ,23289   ,498.3,473.3,441.4
XS GIS Cut Line= 5
2237866.66539132516940.3728526092237830.85900104 517032.33832134
2237742.76470626517177.064662767  2237544.552543517389.434837686
2237483.99435309517626.137077423
#Sta/Elev= 30
       0 2912.98     109 2906.06   284.7 2902.22   295.4 2900.32     323 2890.26
   328.5 2889.23   383.2 2888.03   400.2 2885.05   432.4 2884.05   453.6 2882.82
   465.3 2882.84   471.2 2884.11   477.1 2885.55     509 2884.16   518.1 2884.91
   535.7 2894.61   541.7 2895.61     579  2892.1   587.3 2897.05   595.5 2909.12
   598.2 2912.06     612  2923.1     641 2937.65     674 2957.78   690.9 2973.97
   698.7    2980   727.6 2993.72     740 3000.98   765.8 3011.96   802.9 3023.78
#Mann= 7 ,-1,0
       0     .06       0      10     .05       0  418.12     .07       0
   432.4    .045       0   471.2     .07       0  488.12     .06       0
  608.62      .1       0
Bank Sta=432.4,471.2
XS Rating Curve= 0 ,0
Exp/Cntr=0.3,0.1

Type RM Length L Ch R = 1 ,22815   ,474.5,471.8,464.7
XS GIS Cut Line= 4
 2237267.6847594516555.6852620772237195.32158869516783.786561064
2237281.84277106517376.8499384322237341.62104252517581.354551317
#Sta/Elev= 30
       0 2918.57   165.2 2907.47   211.1 2902.99   232.4 2897.44   256.9 2882.21
   260.9 2881.19   317.5 2877.89   337.7 2879.53   471.1  2882.1   507.5  2881.8
  517.69 2880.18     550 2880.15   568.1  2881.5   657.1 2881.36   673.2 2880.47
   725.8 2881.55   770.4 2878.85   786.4 2881.51   802.6 2880.44   814.7 2881.26
   826.9 2886.53   859.8 2884.58     864 2886.31   880.7 2903.19     889 2909.88
   930.7 2931.94   947.3 2944.52   959.8 2952.72    1018 2980.571051.708 2992.89
#Mann= 9 ,-1,0
       0     .08       0      50      .1       0   309.3     .05       0
  517.69    .045       0     550     .05       0   599.3      .1       0
   699.3     .05       0   799.3     .07       0  898.65      .1       0
#XS Ineff= 2 , 0
          334.88 2896.88
Permanent Ineff=
       F       F
Bank Sta=517.69,550
XS Rating Curve= 0 ,0
Exp/Cntr(USF)=0,0
Exp/Cntr=0.3,0.1

Type RM Length L Ch R = 1 ,22343   ,278,278.5,277.6
XS GIS Cut Line= 4
2236632.14734705516525.7961263482236787.88547532 517175.49155036
2236888.56466936517491.6871441292237171.72490258517650.571497216
#Sta/Elev= 30
       0  2971.5    36.4 2964.12    69.3 2955.34    85.8 2948.74    98.1 2938.76
   106.3 2928.89   142.2 2904.55   155.5 2891.85   168.7 2875.19   172.1 2872.32
   176.2 2871.85   221.5  2873.9   447.7 2874.04   525.9 2876.57     641 2875.59
   679.2  2878.6   699.3 2874.62   771.6  2874.9   806.6 2874.99   879.8 2876.94
   976.3 2875.55   988.9 2880.22  1057.7 2880.78    1105 2885.93  1123.3 2890.86
  1146.3 2894.51  1187.5 2914.09  1260.9 2943.59  1289.1 2958.011324.628 2972.49
#Mann= 10 ,-1,0
       0      .1       0     230     .05       0   738.1    .025       0
   771.6    .045       0   806.6    .025       0   838.1      .1       0
   948.1     .06       0 1079.94     .05       0 1089.94     .07       0
 1199.94      .1       0
#XS Ineff= 2 , 0
          393.02 2889.27
Permanent Ineff=
       F       F
Bank Sta=771.6,806.6
XS Rating Curve= 0 ,0
Exp/Cntr(USF)=0,0
Exp/Cntr=0.3,0.1

Type RM Length L Ch R = 1 ,22065   ,422.8,418.5,405.8
XS GIS Cut Line= 4
2236347.33617299 516561.541215572236353.62862262516712.560006624
2236628.92329381517574.6256055552236699.71335212517911.271660613
#Sta/Elev= 30
       0 2945.43    15.7 2942.76   139.8 2900.89   151.8 2891.09   179.1 2877.34
   202.2 2867.22   214.8 2865.99   235.8 2869.02   349.2  2872.1   449.9 2872.59
   479.3 2870.55   630.5 2874.07   685.1 2870.89   698.6 2868.11   720.2 2870.14
   785.9 2868.94   802.6 2871.62   850.7    2871   882.7  2871.1   920.7 2874.34
  1008.4 2876.54  1058.7 2880.91  1075.1 2876.24  1091.3  2879.5  1291.7  2885.3
  1316.2 2886.95  1332.6 2894.55  1358.2 2887.88  1381.6 2897.811400.114 2899.19
#Mann= 8 ,-1,0
       0      .1       0  201.15     .05       0  601.15     .08       0
   850.7    .045       0   882.7     .08       0  911.15     .05       0
 1021.15     .07       0 1116.11     .05       0
#XS Ineff= 2 , 0
           358.8 2878.97
Permanent Ineff=
       F       F
Bank Sta=850.7,882.7
XS Rating Curve= 0 ,0
Exp/Cntr(USF)=0,0
Exp/Cntr=0.3,0.1

Type RM Length L Ch R = 1 ,21646   ,360.6,387.5,408.7
XS GIS Cut Line= 4
2235854.95198966516825.8240999142236131.81977326517225.394651244
2236320.59326208517613.9534157262236312.72770004 517952.17258319
#Sta/Elev= 30
       0  3022.5    29.2 3005.17      78 2962.88   149.6 2913.67   163.7 2889.83
   169.5  2883.4   184.4 2875.36   193.9 2868.13   205.8 2862.81   223.1 2861.57
     262 2865.84   369.1 2867.65   490.3  2866.4   540.1 2868.52     576 2863.61
   583.7 2861.21   601.5 2861.09   619.3 2863.51   662.8 2870.23   933.3  2878.5
   957.3 2877.43  1053.4 2879.29  1101.4 2885.35  1148.5 2888.23  1179.1 2893.16
  1201.4 2898.76  1217.4 2905.38  1229.4 2914.29  1245.4    29161256.418 2923.18
#Mann= 8 ,-1,0
       0      .1       0     270     .05       0     576    .045       0
   619.3     .08       0  726.12     .05       0  836.12     .07       0
 1038.11     .05       0 1238.11      .1       0
#XS Ineff= 2 , 0
          248.84 2873.73
Permanent Ineff=
       F       F
Bank Sta=576,619.3
XS Rating Curve= 0 ,0
Exp/Cntr(USF)=0,0
Exp/Cntr=0.3,0.1

Type RM Length L Ch R = 1 ,21259   ,514.3,507.5,492.8
XS GIS Cut Line= 5
2235598.53466735 516965.831104122235707.07942342517154.604592937
2235812.47795468517340.2318569412235765.28458247517648.561888676
2235796.74683061517920.710335054
#Sta/Elev= 30
       0 3044.78    36.2 3026.18    65.2 3009.39    86.9 2993.89   123.8 2964.38
   197.7 2914.54   205.8 2906.99   211.5 2891.38   216.1 2881.32   228.1 2873.21
   243.7 2859.24   252.9 2858.31   275.9 2859.73   349.5 2859.84   425.8 2862.42
   449.9  2861.2   484.8 2859.06     501 2859.26     505 2861.22   509.1 2864.94
   513.2 2866.44   598.1 2864.98   654.7 2866.14   699.5 2871.57   723.5 2873.22
   865.4 2873.72   930.4  2876.6   969.3 2880.77  1001.5    2892  1017.1 2899.14
#Mann= 7 ,-1,0
       0      .1       0  317.76     .05       0   449.9    .045       0
     505     .05       0  631.22     .06       0  731.22     .05       0
  933.14      .1       0
#XS Ineff= 2 , 0
           300.7 2868.76
Permanent Ineff=
       F       F
Bank Sta=449.9,505
XS Rating Curve= 0 ,0
Exp/Cntr(USF)=0,0
Exp/Cntr=0.3,0.1

Type RM Length L Ch R = 1 ,20751   ,368.5,384.2,405
XS GIS Cut Line= 4
2235359.42158152516979.9891157812235312.22820931517230.113988464
2235337.39800782517475.5195239262235254.02305026517760.252869559
#Sta/Elev= 30
       0 3038.31   123.7 2975.85   143.7  2964.8     164 2950.29   188.7 2926.53
   213.2  2910.3   233.2 2892.03   269.7 2863.02   281.7 2856.29   290.1 2855.64
   305.9 2853.93     330 2853.72   344.8 2855.79   358.1 2858.25   366.2 2858.39
   470.7 2857.13   490.8 2859.51   516.5 2858.44   557.1 2859.14   569.6 2861.95
     578 2865.52   598.8 2878.94   606.7 2881.96   665.5 2883.14   673.8 2878.93
     703 2879.48   707.2  2879.7   719.7 2886.16   723.9 2886.83797.9202 2889.07
#Mann= 7 ,-1,0
       0      .1       0   290.1    .045       0   344.8      .1       0
  561.23     .05       0  671.23     .07       0  691.23     .08       0
  771.23     .07       0
#XS Ineff= 2 , 0
                          400.61         2863.87
Permanent Ineff=
       F       F
Bank Sta=290.1,344.8
XS Rating Curve= 0 ,0
Exp/Cntr(USF)=0,0
Exp/Cntr=0.3,0.1

Type RM Length L Ch R = 1 ,20367   ,569.9,544.4,519.2
XS GIS Cut Line= 3
2235068.69060122516877.4969501062234928.38878205517313.488946025
2234940.13569031517613.851135729
#Sta/Elev= 30
       0 3047.07    24.9 3034.18    58.5 3011.63    79.6  2998.8   113.1 2983.33
   134.1 2970.71   159.3 2956.82   180.4 2943.93   201.4 2929.32   225.9 2909.46
   251.8 2880.55     256 2875.26   260.2 2862.16  264.15 2852.57   268.6 2850.24
   283.7 2850.14   293.8 2850.56   308.5 2852.56     319 2854.64   340.3 2853.37
     361 2854.96   365.2    2857   369.4 2860.42   377.8 2861.84   415.7 2861.44
   489.7 2864.09   557.9 2873.79   629.8 2876.74   684.8 2880.47   758.6 2883.58
#Mann= 3 ,0,0
       0      .1       0  264.15    .045       0   308.5      .1       0
Bank Sta=264.15,308.5
XS Rating Curve= 0 ,0
Exp/Cntr=0.3,0.1

Type RM Length L Ch R = 1 ,19823   ,389.9,377.7,366.5
XS GIS Cut Line= 2
2234358.70679105516904.5097793922234611.08641885517656.815135729
#Sta/Elev= 30
       0 3006.74     9.1 2999.37    17.6 2994.89    30.2 2986.27    47.1 2977.66
    59.8 2972.84    76.6 2961.93   123.1 2936.23   182.1 2899.58   190.6 2895.79
     199  2888.9   220.9 2867.27   241.2 2850.11   244.9 2848.11   249.6 2847.11
   301.8 2848.09   321.4 2846.99   329.8 2847.32   338.2 2850.79   363.5 2852.22
   460.6 2851.27   498.6 2852.96     545 2858.09   608.3 2860.53   627.2 2860.07
   646.2 2864.66   692.6  2881.4   730.6  2889.8   743.3 2891.57   793.5 2891.59
#Mann= 4 ,-1,0
       0      .1       0   244.9    .045       0   301.8      .1       0
     770     .08       0
Bank Sta=244.9,301.8
XS Rating Curve= 0 ,0
Exp/Cntr=0.3,0.1

Type RM Length L Ch R = 1 ,19445   ,125.2,137.3,146.1
XS GIS Cut Line= 3
2233950.20452005517116.9480573882234268.09718749517535.988391732
2234281.25730945517702.879547547
#Sta/Elev= 30
       0 2991.26     7.3 2985.19    16.5 2979.01    30.4 2972.01    35.8 2968.16
    47.3 2965.48    61.5 2956.69    85.6 2944.17     176 2889.84   216.2 2859.64
   221.7 2854.25   227.1 2847.39     230 2844.97   246.3 2843.98   266.4    2845
   289.9 2844.77   301.5 2846.83   318.5 2847.39   380.5 2847.54     402 2846.32
   457.2 2845.52   512.9  2851.8   547.2 2850.49   553.2 2851.69   563.3 2855.45
   591.4 2870.49   599.4 2872.13   607.4 2875.25   659.6 2880.98   693.4 2881.78
#Mann= 4 ,-1,0
       0      .1       0     230    .045       0   266.4      .1       0
  625.98     .06       0
Bank Sta=230,266.4
XS Rating Curve= 0 ,0
Exp/Cntr=0.3,0.1

Type RM Length L Ch R = 1 ,19308   ,338.4,342.5,346.9
XS GIS Cut Line= 3
2233916.94756224517179.4134383542234094.49481267517648.249146522
2234161.07503158517714.829365434
#Sta/Elev= 30
       0 2962.31     1.9  2961.1    10.4 2960.17    14.7 2958.89    27.6 2949.29
    70.3 2925.33     100 2904.33   109.4 2900.71   131.1  2885.8     143 2876.33
     159 2865.78   178.5 2848.59   185.8 2846.21   198.6 2845.82   211.7 2842.95
   230.3 2842.43   239.7 2841.61   255.2 2842.41   262.8  2845.2   276.9 2844.84
   288.5 2846.11   345.1 2845.04   365.5 2845.42   410.3 2844.12   442.4 2845.73
   459.6 2849.51   480.9 2857.63   509.4 2863.98   537.6 2872.24   595.5 2874.54
#Mann= 4 ,-1,0
       0      .1       0   230.3    .045       0   255.2      .1       0
     490     .06       0
Bank Sta=230.3,255.2
XS Rating Curve= 0 ,0
Exp/Cntr(USF)=0,0
Exp/Cntr=0.3,0.1

Type RM Length L Ch R = 1 ,18965   ,138.5,147,157.2
XS GIS Cut Line= 2
2233686.69097184517248.7678330542233842.04481596517886.828264288
#Sta/Elev= 30
       0 2978.75    25.1 2966.15    61.2 2942.57    70.4 2940.46    77.7 2936.68
   110.8  2909.4   150.6 2883.46     177 2858.53   185.7 2846.82   190.3 2842.79
   206.3 2839.74   247.4 2843.39   280.4 2843.87     301 2841.46   317.4 2843.61
   346.2 2843.62   383.3 2842.82   406.42839.779   428.6 2838.15   440.9 2838.29
   445.2 2839.65   451.8 2847.63   455.1 2849.04   488.3 2850.77   498.6 2850.01
   506.8 2847.36   535.6 2847.42   554.5 2851.94   597.4 2856.27   656.7 2866.68
#Mann= 5 ,-1,0
       0      .1       0   406.4    .045       0   445.2      .1       0
     500     .08       0     520     .05       0
Bank Sta=406.4,445.2
XS Rating Curve= 0 ,0
Exp/Cntr(USF)=0,0
Exp/Cntr=0.3,0.1

Type RM Length L Ch R = 1 ,18818   ,315.7,331.6,351
XS GIS Cut Line= 4
 2233614.0498096517275.3627623182233606.50887637517465.804296325
2233643.66516217517638.1681776932233632.41795282517891.156309029
#Sta/Elev= 30
       0 2963.71    45.9  2942.2    53.9 2936.77    61.9 2935.68    81.9 2925.15
    99.8 2911.84   154.2 2880.02     178 2862.02     194 2846.39   202.2 2841.73
   214.5 2839.59   263.6 2841.22   271.8  2840.2   296.3 2841.61   312.8 2840.57
   366.5 2841.65   385.9 2841.46   391.6 2839.58     398 2837.78     418 2836.98
   426.8 2839.57     434 2843.97     446 2845.63     466 2846.09     478 2844.46
   502.1 2844.05     538 2844.93   558.1  2849.2   582.1 2850.92   620.2 2857.77
#Mann= 5 ,-1,0
       0      .1       0   391.6    .045       0   426.8      .1       0
  466.91     .06       0  566.91     .05       0
Bank Sta=391.6,426.8
XS Rating Curve= 0 ,0
Exp/Cntr=0.3,0.1

Type RM Length L Ch R = 1 ,18487   ,255.6,254.6,256.9
XS GIS Cut Line= 3
2233523.93935236517303.7616054582233263.84535173517686.677773048
2233227.72118498 517899.29429737
#Sta/Elev= 30
       0 2936.66     6.5 2934.05    16.2 2928.01    25.9 2926.52    30.7 2924.84
      44 2916.26   103.3 2888.34   112.9 2882.58   124.7 2877.45     165 2855.94
   176.5 2845.84   185.5 2843.95   195.1 2843.23   204.8 2839.98   225.5 2835.85
     229 2834.66   241.6 2834.24   262.9 2834.28  269.46 2835.84   277.3 2839.41
   306.3 2837.63   325.7 2837.61   444.3 2839.06   473.5 2841.24   485.7 2838.93
   497.9  2838.2   530.4 2840.65   599.3 2840.39   656.1 2861.66678.5605 2868.94
#Mann= 5 ,-1,0
       0      .1       0   225.5    .045       0  269.46      .1       0
     280     .06       0   512.9      .1       0
#XS Ineff= 2 , 0
                          472.43         2843.67
Permanent Ineff=
       F       F
Bank Sta=225.5,269.46
XS Rating Curve= 0 ,0
Exp/Cntr(USF)=0,0
Exp/Cntr=0.3,0.1

Type RM Length L Ch R = 1 ,18232   ,222.8,244.8,264.8
XS GIS Cut Line= 3
2233264.32157109517248.5407624222233049.16458931517595.851296638
2233001.99047641517873.920404854
#Sta/Elev= 30
       0 2867.31     7.9  2865.9    52.5 2864.81    67.4 2863.19    85.4 2854.97
    90.2 2851.76   104.3 2839.13   108.1 2836.99     111 2836.28   131.3 2835.79
   174.8 2836.85   212.7 2834.68   218.5 2833.98   259.5 2833.91   267.9 2834.62
   273.7 2835.97   278.4 2836.29     294 2835.57   334.8 2837.07   344.2 2836.93
   358.4 2835.08   369.6 2834.86   409.9  2838.4   430.2 2838.11   487.1 2838.94
   580.3 2842.07   592.5 2844.08   628.8 2854.34   657.4 2860.15   690.6 2868.41
#Mann= 5 ,-1,0
       0      .1       0   212.7    .045       0   267.9     .05       0
     340     .06       0  548.55      .1       0
Bank Sta=212.7,267.9
XS Rating Curve= 0 ,0
Exp/Cntr=0.3,0.1

Type RM Length L Ch R = 1 ,17987   ,277.7,253.2,228.7
BEGIN DESCRIPTION:
xs 4
END DESCRIPTION:
XS GIS Cut Line= 4
2233142.05530382517089.0808430352233012.00830351517261.444724403
2232832.41958879517342.9821293622232555.81168336517604.108249039
#Sta/Elev= 30
       0 2868.74    81.4 2866.45   102.7 2854.03   129.9 2852.62   135.4 2851.32
   147.1 2845.82   160.5 2834.73   165.5 2833.19   175.6 2832.56   216.1 2834.06
  243.86 2832.02   255.3 2831.01  274.47 2831.99   302.4 2831.52   348.5 2834.34
   384.8 2834.77   396.9 2834.48   404.6 2832.57     428 2834.42   443.2 2834.47
     452 2836.31   482.8 2835.29   505.4 2833.17   567.7  2831.9   626.1  2834.5
   661.1 2834.03   732.5 2836.21   743.5 2837.91   779.9 2858.34793.5451 2867.19
#Mann= 6 ,-1,0
       0      .1       0  243.86    .045       0  274.47      .1       0
  405.92     .06       0  433.15     .05       0  563.15      .1       0
#XS Ineff= 2 , 0
                          518.27         2841.22
Permanent Ineff=
       F       F
Bank Sta=243.86,274.47
XS Rating Curve= 0 ,0
Exp/Cntr(USF)=0,0
Exp/Cntr=0.5,0.3

Type RM Length L Ch R = 1 ,17734   ,42.9,39.6,40.3
BEGIN DESCRIPTION:
xs 3
END DESCRIPTION:
XS GIS Cut Line= 6
2232881.35168834516801.058464474 2232870.2048026517030.675207452
2232816.56375904517120.8630808412232754.32698032517130.009379264
2232684.42337358517097.3798437592232350.94570849517272.014387038
#Sta/Elev= 30
       0 2869.09    62.9  2857.5    94.6 2848.16   110.8 2841.12   147.1 2840.88
   163.1 2837.61   183.3 2836.08   244.7 2835.73   253.6 2831.67   256.4  2830.8
   271.3 2829.62   297.9 2830.69   317.2 2834.64     334  2834.7   364.1 2834.43
   385.6 2832.59     447 2833.17   495.3 2832.52   503.9 2830.53   524.9 2831.59
   553.8 2830.34     587  2829.2   644.5 2828.24   675.7 2830.56   721.6 2828.42
   748.8 2830.56   761.4 2835.51   780.5 2845.92   793.6 2850.99859.0234 2883.97
#Mann= 7 ,-1,0
       0      .1       0   253.6     .05       0   256.4    .045       0
   297.9     .05       0     334      .1       0   553.8     .06       0
     587      .1       0
#XS Ineff= 3 ,-1
       0   243.1 2836.93   311.3     530 2831.24     530 859.023 2837.06
Permanent Ineff=
       F       F       F
Bank Sta=256.4,297.9
XS Rating Curve= 0 ,0
Exp/Cntr(USF)=0,0
Exp/Cntr=0.5,0.3

Type RM Length L Ch R = 1 ,17694   ,344.8,370.4,385.5
BEGIN DESCRIPTION:
xs 2
END DESCRIPTION:
XS GIS Cut Line= 6
2232846.98212398516788.9826715872232808.89693103 516907.88278616
2232826.54616678517023.0672721522232793.10550956517089.948586599
2232666.77413783517037.0008793282232332.36756559517200.488536865
#Sta/Elev= 30
       0  2865.5      59 2852.93    69.2    2849      80 2841.53   104.2 2840.84
   126.1 2835.13   166.2 2834.78   194.5 2834.43   236.2 2830.28   255.1  2828.9
   258.2 2828.74   283.9 2827.26   291.4 2828.85   317.3 2833.73   356.6 2830.27
   409.6 2832.44   446.4 2831.89   455.7 2830.08   460.7 2828.65   472.1 2830.78
     488 2831.42   503.2 2829.45   513.2 2830.88   620.8 2829.15   703.6 2826.19
     717 2826.91   731.5 2830.81   774.8 2850.59   814.9 2864.55832.5097 2872.62
#Mann= 11 ,-1,0
       0      .1       0      80     .07       0   166.2     .05       0
   236.2      .1       0   255.1     .05       0   258.2    .045       0
   291.4      .1       0   455.7     .05       0   472.1      .1       0
   513.2     .06       0   620.8      .1       0
#XS Ineff= 3 ,-1
       0     252  2836.5   297.5     5302830.905     530   789.3 2836.43
Permanent Ineff=
       F       F       F
Bank Sta=258.2,291.4
XS Rating Curve= 0 ,0
Exp/Cntr(USF)=0,0
Exp/Cntr=0.5,0.3

Type RM Length L Ch R = 1 ,17324   ,331.6,331,330.3
BEGIN DESCRIPTION:
xs 1
END DESCRIPTION:
XS GIS Cut Line= 3
2232878.42872618516630.8611155062232675.90896482516764.986156561
2232194.17503137517116.259631486
#Sta/Elev= 30
       0 2886.62   103.5  2866.8   122.6 2860.84     137 2852.19   156.3 2851.96
   180.2 2842.44   218.6 2833.38   257.4 2830.43   311.9 2831.31   383.1 2828.02
     401 2826.52  409.08 2824.13   415.8 2821.97   433.3 2821.56   445.5 2821.91
   451.8 2824.23   460.4 2828.71   478.5 2829.35   494.4 2828.94   509.9 2826.21
   569.3 2827.88   633.7 2825.78   653.5 2823.68   673.3 2830.95   737.6 2874.98
   752.4 2882.57     797  2910.2   812.6 2918.25   831.7 2925.27   839.1 2930.17
#Mann= 6 ,-1,0
       0      .1       0     210     .05       0  382.91     .06       0
  409.08    .045       0   451.8     .06       0  552.91      .1       0
#XS Ineff= 2 , 0
          307.04 2836.13  474.36         2832.78
Permanent Ineff=
       F       F
Bank Sta=409.08,451.8
XS Rating Curve= 0 ,0
Exp/Cntr=0.3,0.1

Type RM Length L Ch R = 1 ,16993   ,309.7,328.5,343.4
XS GIS Cut Line= 2
2232637.68233333516375.0745154082232133.09079772516757.340830263
#Sta/Elev= 30
       0 2865.48     5.4 2864.91      30 2856.55    82.5 2834.88    97.2 2830.77
   179.6 2828.65   202.4 2824.89   217.7 2823.74   242.8 2825.15   338.1 2826.69
   353.2 2825.42   359.5 2821.86   363.2 2820.18   393.3 2819.97   399.5 2820.47
   403.4 2822.13   420.8 2827.45   450.8 2827.28   476.5 2823.61   488.7 2825.23
   503.7 2824.89   513.8 2827.22   523.8 2833.34   539.4 2845.58   559.9 2865.55
     569    2876   573.6 2884.51   579.3 2892.71     605 2910.01633.0404 2925.12
#Mann= 6 ,-1,0
       0     .06       0      20     .05       0     270      .1       0
   359.5    .045       0   403.4     .06       0     510      .1       0
#XS Ineff= 2 , 0
          334.88 2833.48  433.97         2832.69
Permanent Ineff=
       F       F
Bank Sta=359.5,403.4
XS Rating Curve= 0 ,0
Exp/Cntr(USF)=0,0
Exp/Cntr=0.3,0.1

Type RM Length L Ch R = 1 ,16665   ,421.3,393.6,348.6
XS GIS Cut Line= 3
2232515.35711258516241.2813052092232083.39617679516343.218989171
 2231931.7638719516505.045062459
#Sta/Elev= 30
       0 2846.69    60.8 2830.26     106 2828.78   115.6 2827.62   134.8 2823.44
   159.4 2822.35   221.1 2822.34   245.8 2820.25   274.5 2821.67   307.4 2821.99
   316.4 2819.47   323.8  2818.2   340.3 2818.11   364.9 2818.25  370.36  2819.5
   377.3 2821.66   417.5 2822.97   434.8 2826.16   473.9 2823.09   481.5 2827.94
   506.8 2849.78   512.6  2855.6   518.7 2864.42   526.7 2872.28   549.4 2893.09
   556.1 2897.59   577.2  2908.5     589 2912.72   622.9  2929.7665.5917 2942.98
#Mann= 8 ,-1,0
       0      .1       0      60     .05       0      90      .1       0
     290     .05       0   316.4    .045       0  370.36     .05       0
     400     .06       0  513.83      .1       0
#XS Ineff= 2 , 0
          217.96 2826.36  437.13         2827.73
Permanent Ineff=
       F       F
Bank Sta=316.4,370.36
XS Rating Curve= 0 ,0
Exp/Cntr(USF)=0,0
Exp/Cntr=0.3,0.1

Type RM Length L Ch R = 1 ,16271   ,461.5,448.4,419.7
XS GIS Cut Line= 3
2232145.83300822515716.3022328082232005.66869277516214.522663169
 2231921.5701035516489.754409865
#Sta/Elev= 30
       0 2864.84   154.7 2850.58   171.3 2844.26   208.7 2819.92   222.6 2818.74
   227.7 2817.24   241.7 2815.82   266.8 2817.16   310.1 2818.84     379 2818.92
   420.6 2817.12   443.1 2817.52   470.5 2815.52   482.9 2816.17   503.7 2822.16
   552.9 2820.48     558 2820.66   570.5 2824.33   574.7 2824.47   608.2  2821.5
   612.4 2823.62   637.5 2845.64   654.2 2865.87   666.7 2871.85   675.1 2878.52
   687.5 2885.33     696 2891.34   762.9 2920.53   771.3 2923.06805.3547 2938.91
#Mann= 7 ,-1,0
       0     .05       0      50      .1       0   227.7    .045       0
   266.8      .1       0     460     .05       0  567.56     .06       0
  667.56      .1       0
#XS Ineff= 2 , 0
                          506.26         2823.64
Permanent Ineff=
       F       F
Bank Sta=227.7,266.8
XS Rating Curve= 0 ,0
Exp/Cntr(USF)=0,0
Exp/Cntr=0.3,0.1

Type RM Length L Ch R = 1 ,15823   ,414.4,427.4,439.1
XS GIS Cut Line= 3
2231657.80634625515744.3350958982231676.91966199516057.793474079
 2231792.8737775516415.849588993
#Sta/Elev= 30
       0 2844.72    96.5 2839.03   150.3 2836.89   161.1 2834.95   169.2 2831.99
   193.2 2816.78   209.2 2815.46   233.4 2809.65   249.3 2809.81   265.3 2813.93
   293.9 2812.96   309.4 2814.57   342.8 2811.44   389.1    2812   408.2 2809.27
   414.3 2807.49   422.7 2807.15   435.3  2807.3   443.2 2809.51   452.1 2812.73
   473.2 2812.41   481.6 2816.67   485.8 2817.54   523.6 2813.75   545.3 2814.07
   561.5 2817.24   590.9 2838.88   608.3 2849.84   670.8 2883.89690.4041 2895.78
#Mann= 6 ,-1,0
       0     .05       0     120      .1       0   408.2    .045       0
   443.2      .1       0  524.04     .06       0  624.04      .1       0
#XS Ineff= 2 , 0
          313.52 2818.72  487.44          2819.6
Permanent Ineff=
       F       F
Bank Sta=408.2,443.2
XS Rating Curve= 0 ,0
Exp/Cntr(USF)=0,0
Exp/Cntr=0.3,0.1

Type RM Length L Ch R = 1 ,15395   ,377,358.6,333.9
XS GIS Cut Line= 3
2231315.04088393515762.1741905912231271.71736825516386.542504854
2231415.70434684 516606.98274642
#Sta/Elev= 30
       0  2839.8    59.1    2835    91.2 2820.24   168.2 2819.98   207.5 2815.61
   219.5 2809.52   223.5 2808.81   299.7 2811.74   327.8 2806.23   363.9  2803.8
   371.9 2801.91     396 2801.81     408 2801.85   413.8 2803.94     432 2808.91
   448.1 2808.25   461.2 2805.86   492.2 2807.93   512.2 2811.52   552.3 2813.24
   608.5 2811.39   648.1 2812.53   717.7 2810.32   769.7 2811.94   781.3  2815.7
   791.5 2822.48   796.2 2827.13   818.8 2839.65   834.5 2846.58889.1682 2877.24
#Mann= 5 ,-1,0
       0      .1       0   363.9    .045       0   413.8      .1       0
     500     .06       0  705.87      .1       0
#XS Ineff= 2 , 0
                          437.75         2813.97
Permanent Ineff=
       F       F
Bank Sta=363.9,413.8
XS Rating Curve= 0 ,0
Exp/Cntr(USF)=0,0
Exp/Cntr=0.3,0.1

Type RM Length L Ch R = 1 ,15037   ,466,450.8,432.8
XS GIS Cut Line= 2
2230777.31960104 515895.967400792231204.18365262516698.726661986
#Sta/Elev= 30
       0 2861.58    10.4 2853.71    42.1 2836.07    55.7 2824.72    59.2 2823.76
    78.4 2823.88    96.5 2818.58   187.1 2811.73   205.2 2808.47   232.4 2807.64
   261.7 2799.88   300.4 2801.35   337.2 2800.38   350.2 2799.25   381.9 2800.31
     391 2804.59   409.1 2803.28   454.4 2805.71     494 2804.22   529.5 2807.97
   585.4 2807.56     630 2809.05   670.6 2809.73   685.5 2807.25   739.8 2808.93
   804.5 2808.11   830.4 2811.17   851.8 2817.83   880.3 2821.03   909.2  2833.1
#Mann= 6 ,-1,0
       0      .1       0   337.2    .045       0   381.9      .1       0
     630     .06       0     740     .05       0     860      .1       0
#XS Ineff= 2 , 0
                          395.49          2809.9
Permanent Ineff=
       F       F
Bank Sta=337.2,381.9
XS Rating Curve= 0 ,0
Exp/Cntr(USF)=0,0
Exp/Cntr=0.3,0.1

Type RM Length L Ch R = 1 ,14586   ,270.1,291.5,304.6
XS GIS Cut Line= 3
2230383.58529673516306.2665787352230772.22271684516612.079630619
2230944.24255852516883.488714166
#Sta/Elev= 30
       0 2883.25    57.8 2873.97    73.7 2868.37    93.6 2867.58   101.7 2865.71
   134.1 2852.46     160 2840.09   170.6 2836.49   189.1 2825.04   207.6 2815.21
   224.6 2802.34   229.8 2799.83     257 2796.82   280.7 2798.41   290.9 2795.49
   301.1 2794.33   346.9 2793.57   358.6 2795.45   366.9 2799.91   372.8 2800.88
   412.7 2800.51   489.8  2804.6   515.6 2804.09   524.2 2805.53   715.6 2813.67
   737.4 2812.25   775.2 2813.89   789.4  2822.3   794.2 2823.94815.8619 2825.35
#Mann= 7 ,-1,0
       0      .1       0   290.9    .045       0   358.6      .1       0
     400     .07       0     480     .06       0  544.53     .05       0
  654.53      .1       0
Bank Sta=290.9,358.6
XS Rating Curve= 0 ,0
Exp/Cntr(USF)=0,0
Exp/Cntr=0.3,0.1

Type RM Length L Ch R = 1 ,14294   ,180.2,194.5,206.8
XS GIS Cut Line= 2
2230287.49730677516450.8337101742230592.64330393 516985.88422575
#Sta/Elev= 30
       0  2867.1    16.9 2867.45    21.1 2865.96    31.5 2860.16    43.3 2856.38
    62.6  2848.4    98.3 2831.73   138.6 2805.88   154.7 2797.63   196.1    2794
   251.4 2795.16   263.2 2791.99   283.7 2789.85   297.4 2789.79   311.2 2790.21
   316.3 2792.03   324.3 2797.96   332.4 2798.96     357 2799.69   366.5 2798.31
   388.9  2800.2   415.7  2800.9   465.5 2800.14   490.8  2803.1   521.3 2804.46
   527.6 2805.82   536.9 2809.82   569.1  2828.1   587.5 2832.53 615.949 2836.69
#Mann= 6 ,-1,0
       0      .1       0   263.2    .045       0   316.3      .1       0
     340     .06       0     460     .05       0     560      .1       0
Bank Sta=263.2,316.3
XS Rating Curve= 0 ,0
Exp/Cntr(USF)=0,0
Exp/Cntr=0.3,0.1

Type RM Length L Ch R = 1 ,14100   ,130.9,128.3,125.7
BEGIN DESCRIPTION:
xs 4
END DESCRIPTION:
XS GIS Cut Line= 2
2230203.05964728516446.6536280212230292.51340535517049.421474475
#Sta/Elev= 30
       0 2873.59    10.6 2872.18    14.7 2870.63    22.8 2865.93      43  2865.4
    55.1 2859.49    87.1 2847.85   103.6 2842.68   147.6 2824.06   172.2 2810.81
   208.8 2794.79   232.1 2793.32   269.4 2793.52   293.7 2790.08   305.8 2791.05
   310.3 2789.99     318 2787.61   338.2  2787.9   343.6 2790.05   350.3 2794.38
   354.4  2795.3   366.5 2795.31   398.8  2797.7   408.1 2796.94   415.2 2797.87
   463.5  2799.6   564.6 2805.55   580.7 2809.46     597 2816.91609.3694 2821.23
#Mann= 6 ,-1,0
       0      .1       0     310     .07       0   310.3    .045       0
   343.6     .07       0     410     .05       0     510      .1       0
Bank Sta=310.3,343.6
XS Rating Curve= 0 ,0
Exp/Cntr(USF)=0,0
Exp/Cntr=0.5,0.3

Type RM Length L Ch R = 1 ,13971   ,47.2,47.5,48.4
BEGIN DESCRIPTION:
xs 3
END DESCRIPTION:
XS GIS Cut Line= 6
2229935.18827869516620.6244671442230050.06864048516664.853916404
2230078.79427798516680.8763972582230101.56510606516706.353659068
2230112.28441825516736.3083535552230182.15923651517035.209195155
#Sta/Elev= 30
       0 2810.93    21.9 2805.72    32.1 2804.11    46.9 2803.49    52.5 2802.43
   111.6 2798.91   127.8 2799.07   139.3 2796.88   190.6 2793.21   222.1 2792.73
   242.7  2793.9   249.3 2793.28   251.7 2792.14   255.8 2788.07   259.9 2786.06
   269.3 2785.96   284.6 2786.52   288.7 2788.09   296.9  2792.5     301 2793.25
   325.7 2793.93   345.9 2795.49   362.6 2796.12     375 2795.04   444.8 2795.93
   459.3 2796.37   479.1  2799.2   506.4 2801.65   518.3 2807.21     529 2814.01
#Mann= 6 ,-1,0
       0      .1       0   242.7     .07       0   255.8    .045       0
   288.7     .07       0   345.9     .05       0   444.8      .1       0
#XS Ineff= 4 ,-1
   86.54     240 2796.46     240   243.8  2793.1   300.7  361.01 2793.26
  361.01     529 2797.25
Permanent Ineff=
       F       F       F       F
Bank Sta=255.8,288.7
XS Rating Curve= 0 ,0
Exp/Cntr(USF)=0,0
Exp/Cntr=0.5,0.3

Type RM Length L Ch R = 1 ,13924   ,173.5,175.4,177.2
BEGIN DESCRIPTION:
xs 2
END DESCRIPTION:
XS GIS Cut Line= 6
2229902.67392767 516629.741226322229939.71447164516648.133587792
 2230004.0877368516677.3941628632230046.72457476516704.146688642
 2230064.2809198516732.5712472822230129.49020139 517042.73334303
#Sta/Elev= 30
       0 2808.93    69.7 2800.24   101.9 2798.64   111.5 2797.22   121.6 2797.35
   190.4 2792.96   193.3 2792.25   200.5 2787.93   216.5  2789.7     225 2788.94
   233.2 2789.35  235.58 2788.01   241.4 2785.85   261.8  2785.7   265.9 2786.02
   270.5 2787.96   274.1 2790.03   278.2 2791.34   286.4 2792.85   319.1 2793.57
   327.2 2794.72   347.7 2795.52   375.2 2793.87   384.5 2793.98   392.6 2794.93
   417.2 2794.23   449.9 2794.95   482.6 2798.88   490.7 2801.53512.7539 2814.12
#Mann= 6 ,-1,0
       0      .1       0   216.5     .07       0  235.58    .045       0
   270.5     .07       0   319.1     .05       0   417.2      .1       0
#XS Ineff= 3 ,-1
       0   228.5 2792.75   277.5  349.52 2792.75  349.52  502.99 2796.04
Permanent Ineff=
       F       F       F
Bank Sta=235.58,270.5
XS Rating Curve= 0 ,0
Exp/Cntr(USF)=0,0
Exp/Cntr=0.5,0.3

Type RM Length L Ch R = 1 ,13749   ,297.9,298.6,299.6
BEGIN DESCRIPTION:
xs 1
END DESCRIPTION:
XS GIS Cut Line= 2
2229868.26311982516615.6353068682229957.43820575517084.733415142
#Sta/Elev= 30
       0 2812.46    13.8 2811.56      26 2803.53    34.1 2795.97    42.3 2791.66
    62.6 2791.28    74.9 2792.22   123.7 2793.39   144.1 2792.68   164.4 2790.28
   192.3 2791.64   205.2 2786.81   209.2 2785.58   213.4 2785.25   237.7 2784.79
   245.9 2785.02   256.5 2786.69   262.2 2787.85   270.3 2788.29   278.4 2791.63
   281.8 2791.91   306.9 2792.01   319.4 2789.91   372.1 2792.07   392.4  2795.9
   398.1 2796.04   408.7 2797.64   416.9 2800.13   422.1 2802.55477.4989 2832.39
#Mann= 5 ,-1,0
       0      .1       0   205.2    .045       0   256.5      .1       0
     340     .06       0     440      .1       0
#XS Ineff= 2 , 0
          127.89 2798.69  296.62         2796.58
Permanent Ineff=
       F       F
Bank Sta=205.2,256.5
XS Rating Curve= 0 ,0
Exp/Cntr(USF)=0,0
Exp/Cntr=0.3,0.1

Type RM Length L Ch R = 1 ,13450   ,435.2,430.9,426.6
XS GIS Cut Line= 2
 2229579.3729977516604.4884211262229653.68556931517125.605329526
#Sta/Elev= 30
       0 2828.89    24.9 2823.44    32.9 2820.72    41.1 2815.19    61.4 2796.96
      72 2789.87    77.5 2788.24   109.8 2787.67   146.2  2790.1   190.6 2788.41
   210.8 2785.94     235 2787.59   279.5  2787.9   287.8 2787.49   298.4 2783.93
   307.8 2780.67   311.8 2780.53     328 2781.24   333.7 2783.98   340.1 2787.08
   348.2  2792.7   351.4  2793.1   376.5 2793.11   388.6 2790.23   392.6 2791.01
   412.8 2808.81   445.1 2829.27   469.4 2842.65   493.6  2857.8526.3888 2875.72
#Mann= 5 ,-1,0
       0      .1       0   298.4    .045       0   333.7      .1       0
     350     .06       0     450      .1       0
#XS Ineff= 2 , 0
          151.77 2798.22
Permanent Ineff=
       F       F
Bank Sta=298.4,333.7
XS Rating Curve= 0 ,0
Exp/Cntr(USF)=0,0
Exp/Cntr=0.3,0.1

Type RM Length L Ch R = 1 ,13019   ,412.1,414.3,416.9
XS GIS Cut Line= 2
2229162.29368955516793.056571581 2229256.1133112517143.254565283
#Sta/Elev= 30
       0 2821.58    37.6 2817.53    66.4 2812.67    74.7 2810.39    78.8 2808.08
    82.4 2805.14    91.2 2796.15   107.8 2780.59   110.6 2778.71   116.1 2776.81
   132.3 2776.73   140.9 2776.83   148.6 2778.41   161.7 2779.24   165.8 2778.55
   178.2 2778.62   200.9 2785.52     203 2786.36   207.2  2789.6   227.9 2808.12
     232 2810.74   239.1 2813.23   248.6 2814.51   277.6 2814.84   281.7 2817.55
   302.4 2842.22   314.8  2854.3     319 2857.29     338 2867.09362.5476 2878.34
#Mann= 5 ,-1,0
       0      .1       0   110.6    .045       0   148.6      .1       0
     260     .06       0     360      .1       0
Bank Sta=110.6,148.6
XS Rating Curve= 0 ,0
Exp/Cntr(USF)=0,0
Exp/Cntr=0.3,0.1

Type RM Length L Ch R = 1 ,12605   ,409.6,412.8,416
XS GIS Cut Line= 2
2228760.07689572516849.7199074322228842.74963164517232.429651213
#Sta/Elev= 30
       0 2812.94    19.9  2810.3    43.4 2803.76    60.2 2800.81    73.1 2800.22
    81.3 2800.99    89.5 2800.34   101.8 2801.09   109.9 2800.25   138.6 2790.46
   150.9 2787.83   174.6 2773.19   183.6  2770.5   191.4  2770.4   216.3 2770.89
  226.03  2773.2   228.6 2774.02   236.8 2781.22   248.7 2790.31   253.2 2792.23
   277.7 2797.68   302.3 2798.55   310.5 2797.68   314.6 2798.43   322.7 2805.17
   341.5 2816.76   351.4  2819.4   375.9 2833.17   384.1 2835.43391.5374 2838.97
#Mann= 4 ,-1,0
       0      .1       0   174.6    .045       0  226.03     .06       0
     300      .1       0
Bank Sta=174.6,226.03
XS Rating Curve= 0 ,0
Exp/Cntr(USF)=0,0
Exp/Cntr=0.3,0.1

Type RM Length L Ch R = 1 ,12192   ,317.4,320.4,323.3
XS GIS Cut Line= 3
2228367.16151432516905.0515791612228415.45234489517264.012494146
2228452.31292855517393.241085302
#Sta/Elev= 30
       0 2813.21    56.6 2805.74    68.6 2803.41    76.8 2799.87    84.9 2794.48
    92.2 2790.83   104.2 2786.93   143.5 2786.92   153.5 2786.17   157.6 2784.55
   161.6 2782.03   173.7 2772.94  179.74 2769.41   185.8 2767.32     206 2767.06
   226.1 2767.22   232.2 2769.22   242.3 2776.39   258.4 2786.54   266.5  2789.5
   290.7 2790.14   306.9  2789.4     319 2790.34   339.2 2789.46   347.2 2787.86
   351.3 2788.55   363.4  2792.6   413.3 2813.58   475.7 2833.61   496.6 2838.56
#Mann= 5 ,-1,0
       0      .1       0  179.74    .045       0   232.2      .1       0
     240     .06       0     340      .1       0
Bank Sta=179.74,232.2
XS Rating Curve= 0 ,0
Exp/Cntr=0.3,0.1

Type RM Length L Ch R = 1 ,11872   ,329.4,331.5,332.9
XS GIS Cut Line= 3
2228064.54475763 516940.190136292228084.76140123517288.164079919
2228118.37375039517407.830870949
#Sta/Elev= 30
       0 2823.05      13  2820.9      33 2812.49    73.1 2786.11    77.1 2783.83
    81.1 2782.49    89.1 2782.09   101.2 2782.91   133.2 2783.25   152.1 2782.38
   157.3 2780.72   177.3 2767.41   181.3 2765.75   189.3 2763.82   217.4 2763.74
   221.4 2763.84   229.4 2765.83   237.4 2769.81   249.4 2779.82   253.4 2782.37
   257.4 2783.97   305.5 2786.05   329.5 2788.96   337.6 2787.37   345.6 2788.23
   374.5 2787.99   382.9 2789.75   426.8 2792.05   445.2 2794.77   472.9 2800.96
#Mann= 5 ,-1,0
       0      .1       0   181.3    .045       0   229.4      .1       0
  398.56     .06       0  408.56      .1       0
Bank Sta=181.3,229.4
XS Rating Curve= 0 ,0
Exp/Cntr=0.3,0.1

Type RM Length L Ch R = 1 ,11540   ,380.3,375.6,373.8
XS GIS Cut Line= 3
2227741.99466469516949.1129719572227749.42592185517360.618837237
2227810.73379343517520.390866194
#Sta/Elev= 30
       0 2842.03     8.1 2838.72    20.1 2836.97    52.1  2828.2    76.1 2820.41
    88.1 2814.32   100.1 2811.06   120.1 2799.78   135.8 2786.93   148.1 2779.01
   160.1 2773.64   176.1  2770.3   184.1 2764.05   194.8 2762.02   224.1 2761.89
   241.9 2763.76   244.1 2764.43   256.1 2775.87   260.1 2778.43   273.4 2781.23
   328.1 2781.67   375.5 2784.23   404.1 2791.47   433.6 2791.06     455 2788.24
   472.2 2789.36   489.3 2794.06   528.7 2793.87   566.4 2796.99582.7038 2795.94
#Mann= 5 ,-1,0
       0      .1       0   184.1    .045       0   241.9      .1       0
     390     .07       0  491.57      .1       0
Bank Sta=184.1,241.9
XS Rating Curve= 0 ,0
Exp/Cntr(USF)=0,0
Exp/Cntr=0.3,0.1

Type RM Length L Ch R = 1 ,11164   ,414.5,397.9,377.9
XS GIS Cut Line= 3
2227360.21382806517048.5060364832227384.36541383 517344.82741577
2227418.42645704517534.678371105
#Sta/Elev= 30
       0 2817.23     4.7 2813.73    16.7 2806.89    40.8 2789.89    60.9 2779.49
    68.9 2777.99   115.6 2776.59   121.1 2777.58   125.1 2777.06   141.1 2764.88
  151.26 2759.62   161.2 2757.67   193.3 2757.81   197.3  2758.4  200.11 2759.62
   205.4  2763.4   209.4 2768.92   213.4 2772.75   237.5 2790.39   245.5 2793.88
   265.6 2796.62   297.7 2799.55   366.7 2807.37   370.8 2806.14   374.9 2803.93
   407.7 2804.16   411.4 2804.57   419.6 2809.76   423.6 2810.89   490.2 2816.13
#Mann= 5 ,-1,0
       0      .1       0  151.26    .045       0  200.11      .1       0
   397.3     .06       0   447.3      .1       0
Bank Sta=151.26,200.11
XS Rating Curve= 0 ,0
Exp/Cntr=0.3,0.1

Type RM Length L Ch R = 1 ,10766   ,316.7,319.6,321.9
XS GIS Cut Line= 3
2226917.22908624517095.8133862122227077.82605595517372.694630123
2227118.88548568517492.472685239
#Sta/Elev= 30
       0 2850.41     5.9 2849.47    11.9 2846.38    15.5 2843.34    24.7 2833.39
    32.4 2827.95    38.6 2824.89    53.7  2812.4    94.1 2781.91   103.3 2772.91
   117.3 2761.04   127.8 2754.19   131.9 2752.66   140.3 2752.21     168 2752.29
   178.8 2754.04   190.5 2759.72   200.4  2762.4   218.9 2773.19   229.1 2775.65
   237.4 2780.28   243.1 2782.14   283.7 2783.64   292.9 2786.19   308.8  2787.6
     375 2789.17   405.2 2790.81     426  2792.9   435.7 2796.85   446.7 2797.67
#Mann= 4 ,-1,0
       0      .1       0   127.8    .045       0   178.8      .1       0
  390.09     .06       0
Bank Sta=127.8,178.8
XS Rating Curve= 0 ,0
Exp/Cntr=0.3,0.1

Type RM Length L Ch R = 1 ,10447   ,258.4,258.9,259.5
XS GIS Cut Line= 2
2226644.02641918517240.7898155192226783.36249095517517.604144759
#Sta/Elev= 30
       0 2813.42    48.1  2790.6    63.1 2784.69    72.1 2780.28    76.6  2777.6
    85.5 2774.51    94.5 2770.13   101.7 2767.91   112.4 2766.46   116.6 2764.78
   119.6 2762.41   125.8 2756.63   128.5 2754.61   130.3 2753.41   135.8  2751.5
   140.4 2750.21   146.4 2749.37   170.2 2749.16     184 2749.61     193 2751.59
   197.5 2753.27     202 2756.35   211.9 2760.98   224.3 2768.01   228.8 2769.46
   233.3 2770.23   251.2  2771.1   280.4  2778.2   300.5 2780.66309.9044 2780.92
#Mann= 3 ,-1,0
       0      .1       0   135.8    .045       0     193      .1       0
Bank Sta=135.8,193
XS Rating Curve= 0 ,0
Exp/Cntr(USF)=0,0
Exp/Cntr=0.3,0.1

Type RM Length L Ch R = 1 ,10188   ,106.7,109.5,112.2
BEGIN DESCRIPTION:
xs 4
END DESCRIPTION:
XS GIS Cut Line= 2
2226420.28370035 517368.298143532226549.04574253517631.146113631
#Sta/Elev= 30
       0 2790.96    17.9 2780.82    23.3 2778.88    36.6 2772.07    51.4 2766.71
    63.3 2763.56    76.7  2762.8    81.2 2762.08    90.1 2759.07    96.2 2755.71
   107.9 2750.31   116.8 2747.86   123.2 2747.36   130.2 2745.93   143.5 2745.41
   156.9 2745.63  167.76 2747.39   174.7 2748.84   179.1  2750.5   188.1 2755.86
   192.5 2757.53     197 2759.98   205.9 2766.02   210.3 2767.69   214.8 2768.52
   227.8 2769.16   245.3 2770.95   254.7 2771.09   266.7 2772.92   292.7 2773.28
#Mann= 4 ,-1,0
       0      .1       0   123.2    .045       0  167.76      .1       0
     190     .06       0
Bank Sta=123.2,167.76
XS Rating Curve= 0 ,0
Exp/Cntr=0.5,0.3

Type RM Length L Ch R = 1 ,10078   ,41.5,41.8,41.9
BEGIN DESCRIPTION:
xs 3
END DESCRIPTION:
XS GIS Cut Line= 6
 2226220.5509351517439.1726130882226309.53150788517444.048260911
2226328.42464319517447.0955408012226344.27049862517455.627924492
2226359.50689807517481.8345315412226458.84822246517729.273658569
#Sta/Elev= 30
       0 2781.03    15.5  2778.1    96.4 2766.27   159.9 2761.93   169.3 2758.58
   181.4 2757.49   186.2 2756.05   190.6 2751.75   197.6 2747.28   202.9 2745.29
   207.8 2744.53   233.6 2744.44     238 2744.79   244.5 2747.48   250.9 2751.36
   255.2  2755.1   259.5 2756.88   267.5 2758.64   276.8 2763.66   285.4  2767.1
   306.9 2767.68   328.5 2769.45   345.7  2769.6   354.3 2768.75   372.1 2769.42
   381.3  2770.2   390.5 2772.57   406.1 2772.93   414.7 2774.09423.4095 2774.33
#Mann= 5 ,-1,0
       0      .1       0      10     .05       0   197.6    .045       0
   244.5     .05       0  326.77     .06       0
#XS Ineff= 2 , 0
             177 2763.34     254         2764.84
Permanent Ineff=
       F       F
Bank Sta=197.6,244.5
XS Rating Curve= 0 ,0
Exp/Cntr(USF)=0,0
Exp/Cntr=0.5,0.3

Type RM Length L Ch R = 1 ,10037   ,177.4,179.8,182.5
BEGIN DESCRIPTION:
xs 2
END DESCRIPTION:
XS GIS Cut Line= 6
 2226204.0956237517461.1130282932226243.10080629517465.379220138
2226284.54381278517467.2075880722226304.65586006517473.302147851
2226315.62606766517483.0534434972226421.67140781517751.823529751
#Sta/Elev= 30
       0 2779.66    12.2 2778.55    25.5 2776.36    40.3 2775.08    60.4 2771.12
    88.7 2767.06   101.7 2764.32   107.6 2762.47     123 2761.94   135.9 2757.71
   157.4 2755.04   164.7 2752.19     174 2746.89   178.9 2744.96   183.2  2744.5
     209 2744.59   214.1 2745.32  218.52 2746.86   239.1 2756.49     252 2765.19
   256.3 2766.17   273.5 2766.53   290.7 2768.21   312.2 2768.45   320.8 2767.74
   331.2 2768.76   368.1 2768.74   383.7 2770.23   393.9 2772.65405.3553 2773.14
#Mann= 6 ,-1,0
       0      .1       0      30     .05       0     174    .045       0
  218.52     .05       0  276.42     .06       0  386.42      .1       0
#XS Ineff= 2 , 0
           167.4    2763   225.2          2764.5
Permanent Ineff=
       F       F
Bank Sta=174,218.52
XS Rating Curve= 0 ,0
Exp/Cntr(USF)=0,0
Exp/Cntr=0.5,0.3

Type RM Length L Ch R = 1 ,9857    ,343.8,354.5,368.6
BEGIN DESCRIPTION:
xs 1
END DESCRIPTION:
XS GIS Cut Line= 3
2226145.58784982517455.0184685142226147.41621776517531.200465751
2226237.61570249517805.455655807
#Sta/Elev= 30
       0 2783.44     2.2 2781.31    10.2 2774.93    14.2 2772.52    30.2 2765.79
    38.2 2764.28    50.2 2762.89    66.2 2759.34    81.5 2753.85    90.9    2752
   103.6    2752   116.2 2753.04   120.4 2752.78   124.6    2752   138.6 2746.78
   147.1 2745.08   154.4 2743.71   162.5 2743.19   196.2  2743.4  201.75 2745.07
   204.6 2746.38   214.6 2757.82   217.2 2760.39   221.5 2763.13   234.1 2764.27
   267.8 2764.62   283.5 2765.71   347.8 2770.69   360.4 2772.31364.9112 2773.52
#Mann= 4 ,-1,0
       0      .1       0   147.1    .045       0  201.75     .06       0
   286.2      .1       0
Bank Sta=147.1,201.75
XS Rating Curve= 0 ,0
Exp/Cntr(USF)=0,0
Exp/Cntr=0.3,0.1

Type RM Length L Ch R = 1 ,9502    ,317.6,327.7,340.5
XS GIS Cut Line= 4
2225835.06429077517406.1240163552225825.50323102517631.479259295
 2225830.0904268517787.4439157572225880.04818998517905.276782589
#Sta/Elev= 30
       0 2790.93    27.1  2779.2    63.1    2761    75.1 2757.51   103.1 2759.79
   111.2 2759.44   139.2 2754.09   155.2  2753.5     167 2749.49   171.2  2748.9
   191.2 2748.38   211.2 2746.59   231.3 2746.85   235.3 2746.12  244.33 2742.01
   251.3 2740.09   263.3 2740.04   295.3 2740.24   302.9    2742   311.1 2746.45
   323.3 2756.91   327.3 2758.78   339.3 2759.47   343.3 2758.22   351.3 2759.17
   379.3 2759.88   387.8 2764.29   405.2 2768.18   433.3 2772.85   509.6 2782.44
#Mann= 5 ,-1,0
       0      .1       0  244.33    .045       0   302.9      .1       0
  325.56     .06       0  431.59      .1       0
Bank Sta=244.33,302.9
XS Rating Curve= 0 ,0
Exp/Cntr=0.3,0.1

Type RM Length L Ch R = 1 ,9175    ,339.8,339,339.6
XS GIS Cut Line= 2
2225564.53165594517370.0588311312225448.18056095517866.702586811
#Sta/Elev= 30
       0 2788.41    15.5 2786.47    22.9 2784.03    60.7 2759.53    68.9 2756.38
   134.7 2753.61     147 2751.77   196.3 2748.51   212.7 2742.78   229.2 2741.75
   242.5 2738.87   253.8 2736.97   282.1 2736.78   294.9 2736.84  301.34 2738.85
   307.2 2743.75   311.3 2748.61   315.4 2751.71   323.7 2753.47   348.3 2753.92
   364.7 2752.82   385.3 2755.65   393.5 2752.27   430.5 2755.14   446.9 2751.81
   467.4 2752.12   471.6 2752.94   479.8 2756.93   496.2 2767.09   510.1 2771.52
#Mann= 5 ,-1,0
       0      .1       0   242.5    .045       0  301.34      .1       0
     370     .06       0     480      .1       0
Bank Sta=242.5,301.34
XS Rating Curve= 0 ,0
Exp/Cntr=0.3,0.1

Type RM Length L Ch R = 1 ,8836    ,343.1,367.8,387.6
XS GIS Cut Line= 3
2225314.51947124 517196.668677572225192.47021362   517472.074206
2225117.66428601517824.729523485
#Sta/Elev= 30
       0 2786.93    26.8 2781.48    57.4 2778.03    84.8 2773.34   111.3 2767.15
   149.3 2753.22   262.9 2746.22   306.5 2745.58   322.8 2743.24   326.9 2741.48
  333.99 2735.99   339.2 2734.07   367.8 2733.89   379.8    2736   400.5 2738.19
   441.4 2739.95   445.5 2741.24   457.7 2748.91   465.9  2750.6   482.3 2750.88
   501.5 2749.18   531.4 2751.37   547.7 2748.65   562.2 2750.26   580.4 2759.98
   633.6 2795.17   637.7  2798.9   646.5 2813.48   649.9 2815.95   661.7 2820.94
#Mann= 7 ,-1,0
       0      .1       0     180     .05       0     260      .1       0
  333.99    .045       0   379.8      .1       0  471.24     .06       0
  571.24      .1       0
Bank Sta=333.99,379.8
XS Rating Curve= 0 ,0
Exp/Cntr=0.3,0.1

Type RM Length L Ch R = 1 ,8468    ,482.2,474.6,465.8
XS GIS Cut Line= 3
2225142.01106006517170.466083578 2224721.1358474517538.588544785
2224674.11709068517629.185661406
#Sta/Elev= 30
       0 2775.05    14.6 2768.71    31.6 2759.64    40.1 2756.43    76.8 2752.12
     130 2749.17   228.9 2743.81   273.5 2742.89   295.2  2739.2   334.9 2737.37
   350.4 2737.57   362.6 2734.85   374.6 2734.99   388.7 2732.81   397.3 2730.61
   411.4 2730.53   423.3 2731.05  427.94 2732.81   435.5 2742.09   441.6 2745.02
   459.6  2746.5   480.7 2746.55     502 2743.73   544.5 2742.53   553.2 2743.91
   564.8  2748.3   587.3 2759.66   616.1 2770.78   629.7  2774.7661.2228 2789.75
#Mann= 5 ,-1,0
       0     .05       0     130      .1       0   388.7    .045       0
  427.94     .06       0  559.15      .1       0
Bank Sta=388.7,427.94
XS Rating Curve= 0 ,0
Exp/Cntr(USF)=0,0
Exp/Cntr=0.3,0.1

Type RM Length L Ch R = 1 ,7993    ,411.3,386.3,357.9
XS GIS Cut Line= 4
2224787.65018619516878.0323527132224573.19878355517025.969416562
 2224404.6193387517250.7420096982224366.77497353517436.523438718
#Sta/Elev= 30
       0 2762.65    23.7 2760.37    43.1  2757.6    76.7 2755.34   146.4 2748.94
   283.6 2741.25   289.3 2739.74   292.1 2738.12     295 2735.98   299.5 2731.05
   302.2 2729.12   306.4 2728.08   332.1 2727.92   339.5 2727.95   348.9 2729.14
   372.1 2729.45   392.1 2733.34   415.6 2733.21   484.5 2735.99   509.5 2735.66
     515 2736.38   524.5 2739.62   560.3 2737.01   564.4  2738.2   568.5 2740.68
   572.6 2744.23   581.2 2753.85   584.8 2755.99     597 2760.39731.0904 2773.42
#Mann= 7 ,-1,0
       0      .1       0     120     .05       0     170      .1       0
   302.2    .045       0   348.9      .1       0  460.53     .06       0
  530.53      .1       0
#XS Ineff= 2 , 0
                          392.97         2734.84
Permanent Ineff=
       F       F
Bank Sta=302.2,348.9
XS Rating Curve= 0 ,0
Exp/Cntr(USF)=0,0
Exp/Cntr=0.3,0.1

Type RM Length L Ch R = 1 ,7607    ,497.5,494.7,487.3
XS GIS Cut Line= 2
 2224183.2871424516742.7100772542224178.69994662517319.549946372
#Sta/Elev= 30
       0 2841.71    26.5 2828.44    42.5 2822.52    54.5 2814.07    70.5 2805.14
    78.5 2794.47    98.5 2786.86   118.5 2777.44   138.5 2764.78   150.5 2755.55
   154.5 2750.99   166.5 2728.79   170.5  2724.5   182.5 2721.88   198.5 2721.84
   222.5 2722.67   233.2 2724.43   254.5 2726.91   270.5 2726.84   290.5 2732.52
   314.5 2731.23   342.9 2731.88   366.7 2731.04   450.5 2735.56   482.5 2734.24
   498.5 2737.41   518.5 2747.89   526.5 2750.85   554.5 2758.18576.8581 2760.99
#Mann= 5 ,-1,0
       0      .1       0   170.5    .045       0   233.2      .1       0
     400     .05       0     500     .06       0
Bank Sta=170.5,233.2
XS Rating Curve= 0 ,0
Exp/Cntr(USF)=0,0
Exp/Cntr=0.3,0.1
